--- LaurelCrk.prj (project) ---

Proj Title=LaurelCrk
Current Plan=p01
Default Exp/Contr=0,0
English Units
Geom File=g01
Flow File=f01
Plan File=p01
BEGIN DESCRIPTION:
END DESCRIPTION:
DSS Export Rating Curves= 0
DSS Export Rating Curve Sorted= 0
DSS Export Volume Flow Curves= 0
DXF OffsetX= 0
DXF OffsetY= 0
DXF ScaleX= 0
DXF ScaleY= 0

--- LaurelCrk.p01 (plan) ---

Plan Title=Floodplain
Program Version=4.00
Geom File=g01
Flow File=f01
K Sum by GR=0
Std Step Tol=0.01
Critical Tol=0.01
Num of Std Step Trials=20
Max Error Tol=0.3
Flow Tol Ratio=0.001
Split Flow NTrial=30
Split Flow Tol=0.02
Split Flow Ratio=0.02
Log Output Level=0
Friction Slope Method=1
Unsteady Friction Slope Method=2
Unsteady Bridges Friction Slope Method=1
Global Log Level=0
CheckData=False
Run HTab=0
Run UNet=0
Run PostProcess=0
UNET Theta=0
UNET Theta Warmup=0
UNET ZTol=0
UNET ZSATol=0
UNET MxIter=0
UNET MaxInSteps=0
UNET DtIC=0
UNET DtMin=0
UNET MaxCRTS=0
UNET WFStab=0
UNET SFStab=0
UNET WFX=0
UNET SFX=0
UNET DSS MLevel=0
UNET DZMax Abort=0
UNET Convert EG Bridges=0
UNET Use Existing IB Tables=0
UNET Froude Limit=0
UNET Froude Power=0
Write IC File=0
Echo Input=False
Echo Output=False
Write Detailed=0

--- LaurelCrk.f01 (steady flow) ---

Flow Title=NFF Regression Equation
Program Version=4.10
Number of Profiles= 1
Profile Names=P100yr
River Rch & RM=LaurelCrk,Main            ,57026.6
417.3588
River Rch & RM=LaurelCrk,Main            ,56726.6
417.3588
River Rch & RM=LaurelCrk,Main            ,56426.6
539.7373
River Rch & RM=LaurelCrk,Main            ,55826.6
564.1575
River Rch & RM=LaurelCrk,Main            ,53370.4
     606
River Rch & RM=LaurelCrk,Main            ,52978.7
840.4063
River Rch & RM=LaurelCrk,Main            ,52264.8
845.8977
River Rch & RM=LaurelCrk,Main            ,51881.3
989.2965
River Rch & RM=LaurelCrk,Main            ,50229.3
1008.596
River Rch & RM=LaurelCrk,Main            ,49802.3
1119.139
River Rch & RM=LaurelCrk,Main            ,46202.3
1181.804
River Rch & RM=LaurelCrk,Main            ,45218
1312.934
River Rch & RM=LaurelCrk,Main            ,42902.3
1453.656
River Rch & RM=LaurelCrk,Main            ,39217.7
1601.968
River Rch & RM=LaurelCrk,Main            ,36604.6
1766.725
River Rch & RM=LaurelCrk,Main            ,34202.3
1961.884
River Rch & RM=LaurelCrk,Main            ,32082.1
2009.168
River Rch & RM=LaurelCrk,Main            ,28640.9
2225.839
River Rch & RM=LaurelCrk,Main            ,28202.3
2910.688
River Rch & RM=LaurelCrk,Main            ,26952.7
3072.073
River Rch & RM=LaurelCrk,Main            ,22932.1
3365.426
River Rch & RM=LaurelCrk,Main            ,18764.6
 3518.67
River Rch & RM=LaurelCrk,Main            ,10758.9
3892.903
Boundary for River Rch & Prof#=LaurelCrk,Main            , 1
Up Type= 0
Dn Type= 3
Dn Slope=0.025703
DSS Import GetInterval= 0
DSS Import GetPeak= 0
DSS Import FillOption= 0

--- LaurelCrk.g01 (geometry) ---

Geom Title=USGS 10m DEM
Program Version=4.10

River Reach=LaurelCrk       ,Main
Reach XY= 30
     1997345.219      323344.545     1994655.983      321155.309
     1993731.161      321013.218     1993247.667      321109.917
     1992012.679      322604.147     1990065.705      322308.087
     1988444.966      323185.056     1986992.933      323375.762
     1986586.538      323039.287     1986834.854      321659.953
     1984986.266      320646.198     1984669.923      320060.994
     1983496.312      319946.411     1981342.967      318800.288
     1980207.867      319247.006     1977954.645      318423.841
     1977392.146      317854.397     1975755.401      317991.063
     1974355.687      316477.661     1973105.687      313715.508
     1971886.937      312788.425     1970690.756       312562.73
     1970128.257      311630.438     1967496.312      312510.647
      1965019.34       311665.76     1963070.965      311958.563
     1961253.257      309019.328     1958489.368      309232.869
     1956591.358      310445.922       1954658.2         310283.

Type RM Length L Ch R = 1 ,57026.6 ,306.3,299.9,298.9
XS GIS Cut Line= 3
       1997651.4      322893.444     1997337.049      323338.778
     1997077.056      323824.666
#Sta/Elev= 30
       0 2883.35    79.3 2878.13   148.7 2873.14   168.5 2871.25   178.4 2870.54
   188.3 2870.22   198.2 2870.42     218 2871.35   237.9 2871.68   267.6 2871.95
   287.4 2871.78   366.7 2868.98   386.5 2867.69   406.4 2865.95   416.3 2865.44
   537.6 2864.12   545.1 2864.04   552.6 2864.09   643.5 2864.21   653.4 2864.69
   663.2 2865.62   682.9 2868.24   692.7 2869.27   741.9  2873.1   791.1 2875.21
   899.4 2881.29   958.4 2885.05  1007.6 2887.52    1047 2889.11  1096.2 2890.45
#Mann= 3 , 0 , 0
       0      .1       0   537.6    .045       0   552.6      .1       0
Bank Sta=537.6,552.6
XS Rating Curve= 0 ,0
Exp/Cntr=0.3,0.1

Type RM Length L Ch R = 1 ,56726.6 ,291.9,299.8,304.2
XS GIS Cut Line= 3
     1997259.269      322681.566      1997080.33      323198.068
     1996842.294      323699.477
#Sta/Elev= 30
       0 2929.13    99.4 2924.61   119.3 2922.34     169 2914.87   198.8 2910.68
   258.4 2903.06   278.3 2901.07   308.1 2898.59   387.6 2892.94   397.5 2892.03
   407.5  2890.7   427.4 2886.85   506.9 2869.25   526.7 2864.46   536.7 2862.85
   539.1 2862.74   546.6 2862.38   554.1 2862.39   596.2 2862.59     616 2863.12
   645.7 2865.43   665.6 2866.61   774.6 2871.57     834 2875.88   883.6 2878.74
   923.3 2878.79   962.9 2877.29   982.7 2877.04    1062 2878.73  1101.7 2880.04
#Mann= 3 , 0 , 0
       0      .1       0   539.1    .045       0   554.1      .1       0
Bank Sta=539.1,554.1
XS Rating Curve= 0 ,0
Exp/Cntr=0.3,0.1

Type RM Length L Ch R = 1 ,56426.6 ,252.8,246.4,241.1
XS GIS Cut Line= 3
     1997171.864      322628.013     1996825.608      323052.124
     1996497.577      323491.768
#Sta/Elev= 30
       0 2926.23    39.8  2924.7   169.2 2918.09     229 2915.64   248.9 2914.26
   308.6 2908.42   318.6 2906.81   338.5 2902.27   388.2 2888.66   408.1 2884.23
   477.8 2870.12   497.7 2866.37   527.6 2861.36     540 2860.24   547.5 2859.98
     555    2860   567.4 2860.14   577.4 2860.73   617.3 2869.34   627.3 2871.28
   647.2 2874.39   687.1 2878.54     717 2882.76     737 2883.78     757 2883.63
   816.8 2879.95   856.7    2878   956.4 2870.97   966.4 2870.59    1096 2871.16
#Mann= 3 , 0 , 0
       0      .1       0     540    .045       0     555      .1       0
Bank Sta=540,555
XS Rating Curve= 0 ,0
Exp/Cntr=0.3,0.1

Type RM Length L Ch R = 1 ,56180.1 ,354.5,353.6,354.3
XS GIS Cut Line= 3
     1996739.648      322288.846     1996673.044      322817.512
     1996512.779      323190.076
#Sta/Elev= 30
       0 2903.04    69.1 2908.68   108.5 2910.12   197.4 2907.21   236.8 2905.13
   256.6 2903.05   305.9 2896.69   345.4 2892.69   365.1 2889.87   414.4 2880.07
   503.2 2865.63     523 2861.86   552.6 2855.15   562.5 2853.59   572.4 2852.82
   602.1 2852.14   610.1 2851.22   621.9 2850.08   625.1 2850.71   631.8 2852.04
   641.7 2855.24   651.6 2857.34   681.2 2861.98     701 2865.89   780.1 2886.48
   809.8 2892.42   839.5 2895.91   869.2  2898.2   898.8 2899.01   938.4 2898.34
#Mann= 3 , 0 , 0
       0      .1       0   610.1    .045       0   625.1      .1       0
Bank Sta=610.1,625.1
XS Rating Curve= 0 ,0
Exp/Cntr=0.3,0.1

Type RM Length L Ch R = 1 ,55826.6 ,334.7,349.8,363.3
XS GIS Cut Line= 3
     1996530.921      322206.931     1996336.896       322716.65
     1996103.885      323213.832
#Sta/Elev= 30
       0 2901.38    49.6 2892.46    69.4 2890.18    89.2 2885.74   109.1 2882.36
   168.6 2874.13     238 2865.41     357 2846.77   416.5 2834.69   485.9 2818.27
   505.7 2815.23   537.9  2812.3   545.4 2811.44   552.9 2811.32   555.4 2811.28
   585.3 2813.38   635.2 2814.69   675.2 2816.66   705.1 2818.98   735.1 2822.59
     795 2833.71   844.9 2844.32   864.9 2850.07   914.8 2867.15   934.7 2873.48
   954.7 2878.64   994.6 2887.76  1014.6 2891.57  1024.6 2892.92  1094.5 2898.85
#Mann= 3 , 0 , 0
       0      .1       0   537.9    .045       0   552.9      .1       0
Bank Sta=537.9,552.9
XS Rating Curve= 0 ,0
Exp/Cntr=0.3,0.1

Type RM Length L Ch R = 1 ,55476.6 ,238.9,237.7,236.5
XS GIS Cut Line= 4
     1996382.682      322446.262     1996148.668      322471.466
     1995879.359      322631.431     1995692.507        322816.6
#Sta/Elev= 30
       0 2875.76     9.8 2876.69    19.6  2875.5    29.4  2872.3    78.5 2852.05
   107.9 2837.44   166.7 2804.01   186.3 2794.41   196.1 2790.42   215.8  2784.6
   235.4 2780.75   294.8 2773.65   309.8 2773.03   313.7 2772.96   382.2 2775.13
   411.6  2773.5   421.4  2775.4   440.9 2783.22   558.4 2824.05   587.6 2835.96
   636.3 2853.81     646 2858.14   655.8 2863.57     685 2883.02   694.8  2888.8
   704.5 2893.86     724 2901.79   743.5  2907.6   753.2 2908.89   811.7  2910.6
#Mann= 3 , 0 , 0
       0      .1       0   294.8    .045       0   309.8      .1       0
#XS Ineff= 2 , 0
                          357.47         2780.19
Permanent Ineff=
       F       F
Bank Sta=294.8,309.8
XS Rating Curve= 0 ,0
Exp/Cntr=0.3,0.1

Type RM Length L Ch R = 1 ,55238.9 ,252.3,243,230.5
XS GIS Cut Line= 4
     1996331.496      322067.076     1995881.538      322367.047
     1995877.196      322369.942     1995578.039      322729.066
#Sta/Elev= 30
       0 2932.32    40.1 2922.65   130.2 2895.28   160.2 2886.85   170.2 2883.17
   190.3 2871.95   210.3 2857.69   270.4 2810.75   340.5 2753.98   350.5 2748.27
   360.5 2745.92   380.6 2743.47   400.4  2742.1   415.4 2741.74   420.6 2741.69
   460.7 2743.31   500.7 2747.95   520.8 2749.44   555.9 2749.81   595.7 2755.46
   605.7 2758.65   744.9 2813.58   774.7 2826.51   794.6 2836.98   814.5 2848.42
     904 2904.32     914 2910.39   923.9 2915.43   933.8 2918.36  1013.4 2921.52
#Mann= 3 , 0 , 0
       0      .1       0   400.4    .045       0   415.4      .1       0
Bank Sta=400.4,415.4
XS Rating Curve= 0 ,0
Exp/Cntr=0.3,0.1

Type RM Length L Ch R = 1 ,54995.8 ,96.4,95.9,98.8
XS GIS Cut Line= 2
     1995941.643      321877.289     1995615.073      322584.297
#Sta/Elev= 30
       0  2883.2    49.9 2835.35    69.9 2817.94    79.9 2810.04    99.8 2796.43
   109.8  2790.7   129.8  2780.3   159.8 2766.63   179.7 2759.12   199.7 2753.12
   219.7 2748.51   239.6 2744.91   259.6 2742.17   299.5 2738.48   339.5 2735.64
   357.4 2735.75   372.4 2735.82   389.4 2734.95   399.4    2735   429.3 2740.18
   469.3 2742.18   489.2 2744.08   509.2  2747.7   529.2 2753.64   539.2 2758.29
   569.1 2775.76   589.1 2786.05     659 2816.02     669 2821.09   778.8 2897.15
#Mann= 3 , 0 , 0
       0      .1       0   357.4    .045       0   372.4      .1       0
Bank Sta=357.4,372.4
XS Rating Curve= 0 ,0
Exp/Cntr=0.3,0.1

Type RM Length L Ch R = 1 ,54899.9 ,328.8,329,328
XS GIS Cut Line= 3
     1995892.826      321867.189     1995630.223      322293.077
     1995512.388       322550.63
#Sta/Elev= 30
       0 2871.66      10 2863.15      50 2827.67      60 2819.74      80 2806.11
   100.1 2793.63   120.1 2782.42   140.1  2772.5   160.1 2763.68   180.1  2755.9
   200.1 2749.19   210.1 2746.27   240.2 2739.27   300.2 2727.35   330.2  2720.5
   330.6 2720.51   340.2 2720.64   345.6 2721.84   370.2 2728.73   440.3 2744.14
   519.9  2763.1   529.6 2765.94   539.4 2769.88   578.5 2790.44   617.5 2810.37
   637.1 2821.27   715.2 2871.11     764 2903.08   773.8 2908.92   783.6 2912.82
#Mann= 3 , 0 , 0
       0      .1       0   330.6    .045       0   345.6      .1       0
Bank Sta=330.6,345.6
XS Rating Curve= 0 ,0
Exp/Cntr=0.3,0.1

Type RM Length L Ch R = 1 ,54570.4 ,296.3,299.8,302.8
XS GIS Cut Line= 3
     1995600.425      321716.314     1995446.323      321976.038
     1995188.064      322463.829
#Sta/Elev= 30
       0 2791.45     9.7 2783.53    29.2 2770.37   126.6 2711.38   136.4  2705.2
   165.6 2683.95   175.4 2678.54   204.6  2667.4   214.3 2664.48   224.1 2663.05
   233.8 2662.76   294.5 2664.84   309.5 2665.33   341.4 2669.84   380.8 2672.89
   400.6  2675.5   420.3 2679.77     440 2685.91   459.7 2694.79   469.6 2700.72
   518.8 2737.13   538.6 2750.26   558.3 2760.68   617.4 2789.36   656.8 2806.94
   686.4 2816.01   706.1 2820.72     785 2834.83   814.5 2840.94   853.9 2852.77
#Mann= 3 , 0 , 0
       0      .1       0   294.5    .045       0   309.5      .1       0
Bank Sta=294.5,309.5
XS Rating Curve= 0 ,0
Exp/Cntr=0.3,0.1

Type RM Length L Ch R = 1 ,54270.4 ,361.3,376.3,393.9
XS GIS Cut Line= 3
     1995543.173      321414.186     1995181.986      321840.468
     1994865.327      322282.365
#Sta/Elev= 30
       0 2911.53      20 2900.98    49.9 2881.52    69.8  2866.7   139.7 2811.36
   229.5  2749.7   269.4 2724.45   289.3 2713.47   309.3 2703.88   359.2 2683.49
   389.1 2673.69   409.1 2668.67     439 2665.17   518.8 2661.91   551.2 2658.57
   558.7 2657.65   566.2 2657.82   578.5 2660.37   637.8 2684.12     707 2709.77
   736.6 2722.69   766.3 2739.35   776.2 2744.05   894.8 2789.65   954.1 2811.16
   973.9 2816.86   983.8  2818.3  1033.2 2822.38  1052.9  2825.3  1102.4 2839.01
#Mann= 3 , 0 , 0
       0      .1       0   551.2    .045       0   566.2      .1       0
Bank Sta=551.2,566.2
XS Rating Curve= 0 ,0
Exp/Cntr=0.3,0.1

Type RM Length L Ch R = 1 ,53894.1 ,234.7,223.7,212.6
XS GIS Cut Line= 4
     1995091.553       321514.52     1995017.455      321563.455
     1994956.439      321575.936     1994631.814      321632.087
#Sta/Elev= 30
       0 2706.82    29.6 2686.95    39.5 2681.45    49.3  2675.1    59.2 2667.12
    69.1  2658.1    78.9 2649.45    88.8 2642.23    97.7 2638.12   106.6 2635.97
   115.5 2634.68   124.4 2633.81   133.3 2633.33   142.2 2633.26     149 2633.43
     164 2634.11     181 2635.05     191 2635.43     201 2635.55     211 2635.41
     221  2635.9   240.9 2638.97   290.8 2644.31   300.8 2645.94   310.8 2648.37
   320.8 2651.25   360.7 2663.43   450.6 2691.31   460.6 2694.26   480.5 2699.63
#Mann= 3 , 0 , 0
       0      .1       0     149    .045       0     164      .1       0
Bank Sta=149,164
XS Rating Curve= 0 ,0
Exp/Cntr=0.3,0.1

Type RM Length L Ch R = 1 ,53670.4 ,124.9,125.4,121.7
XS GIS Cut Line= 3
     1995306.636      321025.517      1994899.63      321369.122
     1994409.703      321751.738
#Sta/Elev= 30
       0 2828.29    49.3 2824.57   128.2 2815.47   157.8 2814.21   207.1 2814.54
     217 2813.31   226.9 2809.52   246.6 2798.48   266.3 2785.38   295.9 2761.75
   325.5  2733.5   374.8  2683.4   394.6 2665.39   414.3  2649.8     434  2637.3
   453.7 2628.53   473.5 2623.74   503.1 2621.42   525.2 2621.98   540.2 2623.18
     582 2627.42   601.7 2628.07   660.9 2633.03   739.9 2643.54   759.6 2648.62
   868.1 2683.49   917.5  2698.4   937.2 2705.28   986.5 2727.89  1154.3 2818.61
#Mann= 3 , 0 , 0
       0      .1       0   525.2    .045       0   540.2      .1       0
Bank Sta=525.2,540.2
XS Rating Curve= 0 ,0
Exp/Cntr=0.3,0.1

Type RM Length L Ch R = 1 ,53545   ,179.8,174.4,170.5
XS GIS Cut Line= 3
      1995131.95      321045.712      1994820.53      321272.965
     1994473.759      321650.036
#Sta/Elev= 30
       0 2774.98    29.7 2772.16      89 2767.95   108.7 2765.83   128.5 2763.02
   138.4 2760.67   148.3 2757.25     168 2746.47   217.5 2715.36     257 2689.81
   276.8 2677.66   306.4 2660.75   326.2 2650.74     346 2642.03   384.4 2628.62
   399.4 2623.91   405.2 2622.48   415.1 2622.36   434.8 2624.24   474.2  2626.6
   513.6 2630.17   572.7 2638.06   582.6 2639.21   612.1 2641.37     622 2643.12
   799.3  2698.1   809.1 2701.98     819 2706.82   848.6  2723.3   897.8  2752.3
#Mann= 3 , 0 , 0
       0      .1       0   384.4    .045       0   399.4      .1       0
Bank Sta=384.4,399.4
XS Rating Curve= 0 ,0
Exp/Cntr=0.3,0.1

Type RM Length L Ch R = 1 ,53370.4 ,405.1,391.6,379.8
XS GIS Cut Line= 3
     1995000.283      320747.767     1994677.618      321172.241
     1994346.741      321695.331
#Sta/Elev= 30
       0 2681.34    29.6 2673.84    49.4 2670.15    69.1 2667.26   118.5 2661.75
     158 2659.34   177.7 2657.53   207.4 2654.36   227.1 2651.66   256.7 2646.51
     316 2634.94   385.1 2624.12   414.7 2620.91     474 2616.05   503.6 2611.67
   525.7 2610.98   533.2 2610.91   540.7 2611.26   603.1 2616.37     663 2623.79
   742.8 2631.84   752.8 2633.79   762.8 2637.09   852.6 2671.88   872.6 2678.74
   912.6  2690.5   932.5 2699.05   962.5 2714.67  1092.2 2787.53  1152.1 2819.24
#Mann= 3 , 0 , 0
       0      .1       0   525.7    .045       0   540.7      .1       0
Bank Sta=525.7,540.7
XS Rating Curve= 0 ,0
Exp/Cntr=0.3,0.1

Type RM Length L Ch R = 1 ,52978.7 ,207.8,208.3,208.5
XS GIS Cut Line= 2
     1994328.245      320807.363     1994282.622      321561.898
#Sta/Elev= 30
       0 2718.69      10 2711.89   119.4 2643.31   139.2 2631.85   159.1 2621.72
     179 2612.84     189 2608.84   208.9 2602.15   218.8 2599.44   238.7 2595.08
   258.6 2592.24   268.6 2591.53   278.5 2591.56   315.3 2594.67   330.3 2595.26
   427.7 2602.52   437.6 2603.66   447.6 2606.12   467.5 2613.54   507.3 2626.84
   527.2 2634.81     557  2649.2   566.9 2654.71   586.8 2667.08   616.7 2687.04
   636.6 2701.06   686.3 2738.03   706.2 2752.04   726.1 2765.14   755.9 2782.04
#Mann= 3 , 0 , 0
       0      .1       0   315.3    .045       0   330.3      .1       0
Bank Sta=315.3,330.3
XS Rating Curve= 0 ,0
Exp/Cntr=0.3,0.1

Type RM Length L Ch R = 1 ,52770.4 ,299.6,302,301.5
XS GIS Cut Line= 3
     1994153.383      320547.253     1994107.635      321092.927
     1994066.973      321641.673
#Sta/Elev= 30
       0 2851.86    29.9 2846.28    89.6 2833.12    99.6 2830.48   109.5 2826.51
   129.4 2815.48   189.2 2779.17   209.1 2764.98     239 2742.37   258.9 2728.78
   388.3 2653.66   428.1 2632.99   467.9 2614.19   527.7 2589.28   537.6 2588.34
   540.1 2588.43   555.1 2589.14   687.6 2596.37   707.7 2598.39   717.7    2601
   757.7 2616.67   807.7 2637.42   837.7 2648.59   857.7 2657.51   887.7 2673.84
   957.8 2718.43  1017.8  2754.3  1037.8 2765.69  1057.8 2775.33  1097.8 2790.42
#Mann= 3 , 0 , 0
       0      .1       0   540.1    .045       0   555.1      .1       0
Bank Sta=540.1,555.1
XS Rating Curve= 0 ,0
Exp/Cntr=0.3,0.1

Type RM Length L Ch R = 1 ,52468.2 ,214.9,203.8,195.7
XS GIS Cut Line= 3
     1993928.352      320764.592     1993825.668      321003.628
     1993791.569      321602.688
#Sta/Elev= 30
       0  2702.1      50 2671.32      80 2651.78      90 2645.72   100.1 2640.47
   120.1 2631.78   190.1 2605.29   210.1 2598.19   240.2 2588.19   250.2 2584.04
   260.2 2580.42   265.9 2579.84   270.2  2579.4   280.9 2579.27   290.2 2579.25
   300.2 2579.57   310.2  2580.5   360.2 2587.52   390.2 2591.17   400.2  2592.6
   410.2 2594.54   480.2 2612.39   560.2  2633.4   630.2 2653.05   650.2 2659.52
   670.2 2666.67   770.2 2704.53   790.2 2713.15   830.2 2732.54   860.2 2746.32
#Mann= 3 , 0 , 0
       0      .1       0   265.9    .045       0   280.9      .1       0
Bank Sta=265.9,280.9
XS Rating Curve= 0 ,0
Exp/Cntr=0.3,0.1

Type RM Length L Ch R = 1 ,52264.8 ,399.1,382.7,360.9
XS GIS Cut Line= 3
     1993747.055      320624.032      1993570.64      320808.528
      1993736.45      321397.533
#Sta/Elev= 30
       0 2726.24    29.4 2709.55    68.7 2689.13    88.4 2677.65   117.8 2657.89
   127.6  2651.7   157.1 2635.37   166.9 2629.73   176.7 2623.64   196.4 2610.71
   206.2 2603.88   225.8 2588.18   235.6 2582.44   245.4 2580.61   265.1 2579.06
   294.7 2578.36   383.6 2578.01     423 2577.38   462.5 2575.66   511.9 2571.87
   534.8 2570.87   541.5 2570.82   549.8 2571.29   561.2 2573.27   610.6 2587.14
   679.6 2607.61   719.1 2618.72     808 2642.75   847.4 2653.69   867.2 2659.57
#Mann= 3 , 0 , 0
       0      .1       0   534.8    .045       0   549.8      .1       0
Bank Sta=534.8,549.8
XS Rating Curve= 0 ,0
Exp/Cntr=0.3,0.1

Type RM Length L Ch R = 1 ,51881.3 ,297.1,292.1,294.7
XS GIS Cut Line= 4
     1992956.422      320879.215     1993241.373      321061.282
     1993478.663      321241.074     1993662.382        321441.3
#Sta/Elev= 30
       0 2665.73      10 2663.39    19.9  2661.7    29.8 2659.16    69.6 2647.18
    99.5 2637.02     189 2604.99   238.7  2588.1   248.6 2585.65   328.2 2569.35
   348.1 2564.19     358 2562.38   367.9 2561.98   385.8 2562.45   400.8 2563.08
   427.5 2564.22   506.8 2565.79   556.5 2565.44   586.2 2565.98   606.1 2567.55
   645.6 2572.77     665 2575.86   684.4 2580.14   703.8    2586   723.2 2593.15
   781.4 2616.84   810.6 2627.98   839.7 2638.47   868.8  2647.6   907.6 2661.46
#Mann= 3 , 0 , 0
       0      .1       0   385.8    .045       0   400.8      .1       0
Bank Sta=385.8,400.8
XS Rating Curve= 0 ,0
Exp/Cntr=0.3,0.1

Type RM Length L Ch R = 1 ,51589.2 ,293.2,300,303.1
XS GIS Cut Line= 3
     1992657.449      321107.715     1993147.866      321337.143
     1993609.683      321620.096
#Sta/Elev= 30
       0 2726.96    29.5  2713.4   118.1 2676.79     128 2673.34   147.7 2669.11
   157.5 2666.22   295.3 2616.21   344.6 2595.68   354.4 2592.53   374.1    2588
   413.5 2574.62   433.1  2569.2   482.4 2561.56     502 2557.15   511.9  2553.5
   521.7 2548.54   531.6 2544.71   533.9 2544.46   541.4 2543.66   548.9 2544.15
   630.1 2551.61   669.4 2559.18   708.8 2565.09   728.5 2570.32   767.9 2582.67
   817.2 2593.08   836.8  2598.4   866.4  2608.8   984.6 2656.91    1083 2702.38
#Mann= 3 , 0 , 0
       0      .1       0   533.9    .045       0   548.9      .1       0
Bank Sta=533.9,548.9
XS Rating Curve= 0 ,0
Exp/Cntr=0.3,0.1

Type RM Length L Ch R = 1 ,51289.2 ,292.8,300,306.1
XS GIS Cut Line= 3
     1992592.889      321223.487     1993010.999      321601.671
     1993422.512      321940.627
#Sta/Elev= 30
       0 2730.73    29.7 2714.29      89 2678.57   118.7 2661.71   168.1 2630.78
     178 2625.12   187.9 2620.12   197.8 2615.68   207.7 2611.98   227.5 2606.48
   247.3 2602.12   306.6 2590.69     544 2539.77   556.3 2537.56   563.8 2537.06
   571.3 2537.35   583.5 2538.64     623  2544.2   642.8 2548.04   662.5 2552.72
   711.9 2567.34   761.2 2583.92   820.5 2604.89   958.7  2655.8   968.6 2660.09
   978.4  2665.4  1027.8 2695.16  1047.5 2704.96  1077.2 2718.49  1096.9 2728.46
#Mann= 3 , 0 , 0
       0      .1       0   556.3    .045       0   571.3      .1       0
Bank Sta=556.3,571.3
XS Rating Curve= 0 ,0
Exp/Cntr=0.3,0.1

Type RM Length L Ch R = 1 ,50989.2 ,303.9,287.7,274.2
XS GIS Cut Line= 3
     1992528.635      321278.479     1992787.572      321775.101
     1993097.307      322249.472
#Sta/Elev= 30
       0 2742.98      70 2699.21      90 2687.63     120 2671.64     130 2666.88
     150 2658.83     180 2648.71     220    2637     300 2612.03     320  2605.4
     350 2594.58   430.1 2571.82   450.1 2564.92   470.1 2556.99   490.1 2549.82
   510.1  2544.3   530.1 2539.81   540.1 2537.64   552.6 2536.21   560.1 2535.98
   567.6 2536.12   629.6 2538.26   699.2 2542.97   719.1 2545.58   758.9 2552.65
   808.6 2560.69   888.1 2575.96  1027.2 2604.74    1057 2612.59  1126.6 2634.54
#Mann= 3 , 0 , 0
       0      .1       0   552.6    .045       0   567.6      .1       0
Bank Sta=552.6,567.6
XS Rating Curve= 0 ,0
Exp/Cntr=0.3,0.1

Type RM Length L Ch R = 1 ,50701.5 ,291.4,299.3,308.1
XS GIS Cut Line= 4
     1992056.741      321771.358     1992570.742      321935.849
     1992863.338      322048.251     1993038.099      322301.874
#Sta/Elev= 30
       0 2791.91      50 2791.99      60 2791.32      70 2789.03    99.9 2777.28
   139.9 2758.68   169.9 2743.29   219.9 2714.27   299.8 2662.95   319.8  2650.9
   349.8 2634.22   379.8 2615.28   389.8 2609.48   459.7 2572.45   489.7  2555.5
   499.7  2548.7   509.7 2540.51   519.7 2533.89   529.7 2531.92   544.1 2532.33
   559.1  2532.6   686.6 2533.54   735.6 2534.36   755.2 2535.88   853.1 2556.04
   932.6 2570.31  1012.1 2585.43  1081.6 2597.09  1131.3 2607.53  1161.1  2615.7
#Mann= 3 , 0 , 0
       0      .1       0   544.1    .045       0   559.1      .1       0
Bank Sta=544.1,559.1
XS Rating Curve= 0 ,0
Exp/Cntr=0.3,0.1

Type RM Length L Ch R = 1 ,50402.3 ,172.1,172.8,171.7
XS GIS Cut Line= 3
     1992010.636      321846.481     1992452.614      322202.427
     1992845.919      322575.577
#Sta/Elev= 30
       0 2785.72    89.6 2781.75    99.6 2779.76   109.5 2776.19   129.4 2765.34
   159.3 2746.62   209.1 2713.04   248.9 2685.25   288.7 2658.76   308.6 2646.45
   338.5 2630.28   398.2 2602.29   507.8 2542.12   527.7  2529.7   537.6 2524.43
   547.6 2522.33     560 2522.72     575 2524.38   606.9 2527.73   626.6 2528.69
   656.2 2528.71   695.6 2526.42   715.4 2526.91   754.8 2532.74   873.1 2552.12
   912.5 2564.28   981.5 2581.29  1011.1 2589.74  1080.1 2612.09  1109.6 2623.28
#Mann= 3 , 0 , 0
       0      .1       0     560    .045       0     575      .1       0
Bank Sta=560,575
XS Rating Curve= 0 ,0
Exp/Cntr=0.3,0.1

Type RM Length L Ch R = 1 ,50229.3 ,408.7,426.9,443.5
XS GIS Cut Line= 3
      1992102.19       322003.97     1992254.474      322259.408
     1992742.724      322677.635
#Sta/Elev= 30
       0 2733.07    19.8 2717.95    29.7 2711.05    59.5 2691.94   158.6 2632.65
   178.4 2621.63   218.1  2600.7     228 2595.08   267.6 2569.88   277.6 2564.16
   307.3 2549.09   327.1 2540.29   366.6 2524.37   376.5 2520.77   386.4 2519.13
   394.3 2519.14   409.3 2519.44   495.2 2522.99   534.8 2524.13   554.5 2525.34
   574.3 2528.06     604 2533.37   673.2 2540.37   732.6 2548.23   742.5  2550.1
   752.4 2552.65   811.7 2570.05   831.5 2576.28   861.2 2586.84   940.3 2616.49
#Mann= 3 , 0 , 0
       0      .1       0   394.3    .045       0   409.3      .1       0
Bank Sta=394.3,409.3
XS Rating Curve= 0 ,0
Exp/Cntr=0.3,0.1

Type RM Length L Ch R = 1 ,49802.3 ,298.2,299.8,301.3
XS GIS Cut Line= 3
     1991976.614      322031.873     1992014.174      322603.603
     1992084.237      323131.504
#Sta/Elev= 30
       0 2717.85    39.5 2682.29    59.3 2665.15      79 2649.19    98.8 2634.77
   118.5 2622.51   148.2 2606.71   167.9 2597.95   187.7 2590.15   207.4    2584
   237.1 2576.62   296.4  2560.5   414.9 2519.98   424.8 2518.06   434.7 2517.58
   565.5 2515.14     573 2514.97   580.5 2515.08   592.7 2516.28   602.6 2518.81
     642 2531.14   740.6    2572   799.8 2595.25   878.7 2627.42   898.4 2636.65
   967.4 2675.86  1016.7 2701.98  1026.6 2706.11  1046.3 2712.75  1105.5 2729.92
#Mann= 3 , 0 , 0
       0      .1       0   565.5    .045       0   580.5      .1       0
Bank Sta=565.5,580.5
XS Rating Curve= 0 ,0
Exp/Cntr=0.3,0.1

Type RM Length L Ch R = 1 ,49502.3 ,369.3,368.9,369.7
XS GIS Cut Line= 3
     1991817.701      321950.484     1991797.666      322605.454
     1991811.508      323131.895
#Sta/Elev= 30
       0 2715.74    49.6 2697.52    89.4 2680.52   208.5 2610.66   258.1 2585.12
     278 2575.87   287.9 2572.22   347.5 2555.47   407.1 2541.98   466.6 2519.69
   476.6  2517.1   496.4 2515.86   595.7  2515.9   647.8 2514.79   655.3 2514.68
   662.8 2514.68   675.2 2515.47   685.1 2517.92     705 2525.49   744.7 2538.26
   844.1 2576.57   933.5 2612.36   983.2 2633.46    1013 2647.26  1042.8 2663.19
  1102.4 2697.59  1132.2 2717.09  1152.1 2728.85    1172 2737.73  1181.9 2740.59
#Mann= 3 , 0 , 0
       0      .1       0   647.8    .045       0   662.8      .1       0
Bank Sta=647.8,662.8
XS Rating Curve= 0 ,0
Exp/Cntr=0.3,0.1

Type RM Length L Ch R = 1 ,49133.1 ,226.1,230.6,240.2
XS GIS Cut Line= 2
     1991513.365      321982.741      1991541.44      323000.485
#Sta/Elev= 30
       0  2682.5    59.9 2649.95    89.8  2634.4   119.8 2620.53   149.7    2608
   179.7 2598.52   189.6 2596.15   199.6  2595.5   209.6 2595.73   219.6 2594.72
   239.6 2589.94   259.5 2583.72   289.5 2572.05   359.3 2539.22   389.3 2526.87
   409.2 2520.19   419.2 2517.98   439.2 2514.82   479.1 2511.36     496 2510.61
   499.1 2510.55     511 2511.12     549 2516.02   598.9 2524.29   678.8 2536.11
   688.7 2538.56   738.6 2557.76   838.5 2591.08   968.2 2636.62  1018.1 2652.94
#Mann= 3 , 0 , 0
       0      .1       0     496    .045       0     511      .1       0
Bank Sta=496,511
XS Rating Curve= 0 ,0
Exp/Cntr=0.3,0.1

Type RM Length L Ch R = 1 ,48902.3 ,295.2,299.8,296.1
XS GIS Cut Line= 3
     1991410.919      321923.913     1991302.485      322476.098
     1991083.307      322972.869
#Sta/Elev= 30
       0 2715.72    49.4 2676.02    88.8 2639.33    98.7 2632.11   108.6 2626.64
   128.3 2618.02   148.1 2611.21   167.8 2606.84   207.3  2600.5   217.2 2597.17
   246.8 2582.29   296.2 2554.26     306 2549.27   325.8 2541.07   345.5 2534.89
   365.3 2529.86   394.9 2524.46   493.6 2514.17   555.2 2509.73   570.2 2508.34
   572.6 2508.14   582.5 2508.33   592.4 2510.29   641.7 2524.76   839.2 2602.18
   898.4 2624.52   937.9 2640.65   967.5  2653.8  1026.7 2681.38  1105.7 2719.45
#Mann= 3 , 0 , 0
       0      .1       0   555.2    .045       0   570.2      .1       0
Bank Sta=555.2,570.2
XS Rating Curve= 0 ,0
Exp/Cntr=0.3,0.1

Type RM Length L Ch R = 1 ,48602.3 ,411.4,403.8,399.6
XS GIS Cut Line= 3
     1991249.662      321879.595     1991021.194       322381.23
     1990886.341      322906.899
#Sta/Elev= 30
       0 2708.34    29.5 2689.15    88.6 2652.12   137.8 2620.46   147.6 2615.25
   157.5 2611.42   167.3  2608.6     187 2604.56   246.1 2597.59   265.8  2592.9
   305.1 2580.25   403.6 2549.98   433.1 2538.85   472.5 2523.03   492.2 2516.07
   531.5 2506.12   543.7  2503.8   551.2  2503.2   558.7 2503.78   600.6 2510.31
   620.3 2514.49   630.2 2517.33     788 2572.62   807.8 2578.29   827.5 2582.74
   847.2    2589     867 2598.34   916.3 2625.11   985.4 2661.73  1093.9 2714.64
#Mann= 3 , 0 , 0
       0      .1       0   543.7    .045       0   558.7      .1       0
Bank Sta=543.7,558.7
XS Rating Curve= 0 ,0
Exp/Cntr=0.3,0.1

Type RM Length L Ch R = 1 ,48198.3 ,192,196.1,200.7
XS GIS Cut Line= 2
     1990680.109      321840.549     1990612.603      322874.144
#Sta/Elev= 30
       0 2613.89    29.9  2606.3    49.8 2600.81    79.7 2591.41    99.6 2583.93
   129.5 2569.73   139.4 2566.19   169.3 2558.15   219.1 2546.84     239 2542.85
   318.7 2528.27   368.5 2519.71   517.9 2505.66   527.9 2504.21   537.8 2501.83
   545.1 2499.48   557.7  2496.1   560.1 2496.13   567.7 2496.22   577.7 2499.13
   607.5 2511.58   647.4 2530.46   687.2 2546.93   717.1 2557.94     747  2567.3
   916.3  2630.8   926.2    2635   966.1 2654.59  1005.9 2671.76  1035.8 2684.04
#Mann= 3 , 0 , 0
       0      .1       0   545.1    .045       0   560.1      .1       0
Bank Sta=545.1,560.1
XS Rating Curve= 0 ,0
Exp/Cntr=0.3,0.1

Type RM Length L Ch R = 1 ,48002.3 ,307.3,299.9,292.6
XS GIS Cut Line= 3
     1990582.809      321830.164     1990451.157      322360.266
     1990306.392      322886.688
#Sta/Elev= 30
       0 2657.51    29.8 2647.56   109.2 2615.49   168.8 2592.76   278.1 2555.11
   297.9  2547.8   337.6 2532.15   377.4  2514.7   387.3    2512   397.2 2510.91
   506.5 2500.58   516.4 2498.85   538.7 2491.11   546.2 2489.17   553.7 2489.15
   556.1 2489.14   566.1 2491.75   585.9 2500.31   615.7 2509.69   665.3 2522.96
   744.7 2545.37   804.3 2560.59   824.2 2566.63   863.9 2580.02   883.7 2587.46
   923.4 2603.72  1002.8 2637.86  1042.5 2652.68  1072.3 2669.06  1092.2 2676.47
#Mann= 3 , 0 , 0
       0      .1       0   538.7    .045       0   553.7      .1       0
Bank Sta=538.7,553.7
XS Rating Curve= 0 ,0
Exp/Cntr=0.3,0.1

Type RM Length L Ch R = 1 ,47702.3 ,305.4,300,293.5
XS GIS Cut Line= 3
      1990109.58      321758.135     1990157.124      322306.351
     1990189.198      322865.267
#Sta/Elev= 30
       0  2678.7      60 2656.07   160.1 2615.55   180.1 2608.25   220.1 2594.56
   270.1 2574.71   320.2 2555.97   380.2 2536.21   390.2 2533.25   430.2  2523.2
   470.2 2514.27   480.2 2510.89   490.2 2506.68   530.3 2488.88   540.3 2486.49
   542.8 2486.48   550.3 2486.46   557.8 2487.52   580.3 2491.22   630.2  2498.2
   700.2  2507.1   740.2 2512.56   750.2 2514.42   770.2 2519.55   830.2 2537.63
   900.2 2560.82   920.2 2568.08  1000.1 2598.52  1050.1  2618.4  1110.1 2640.74
#Mann= 3 , 0 , 0
       0      .1       0   542.8    .045       0   557.8      .1       0
Bank Sta=542.8,557.8
XS Rating Curve= 0 ,0
Exp/Cntr=0.3,0.1

Type RM Length L Ch R = 1 ,47402.3 ,305.3,300,293.8
XS GIS Cut Line= 3
     1989699.212      321868.889     1989874.981      322390.884
     1990057.285      322904.653
#Sta/Elev= 30
       0 2755.07      20 2747.93      30 2743.64    40.1 2738.22   100.1 2698.01
   140.2 2674.42   350.5 2564.82   360.5 2559.35   390.6 2540.61   400.6 2536.33
   410.6  2533.2   430.6 2528.11   450.6 2524.76   460.7 2521.67   470.7 2515.66
   480.7 2508.68   500.7 2493.04   510.7 2486.97   520.8 2484.32   530.8 2484.21
   543.3 2485.44   558.3  2487.1   699.5 2501.68   739.1 2506.32   758.9  2509.8
   887.8 2548.48   937.4 2565.62  1016.6 2596.09  1046.4 2608.88    1096 2631.39
#Mann= 3 , 0 , 0
       0      .1       0   543.3    .045       0   558.3      .1       0
Bank Sta=543.3,558.3
XS Rating Curve= 0 ,0
Exp/Cntr=0.3,0.1

Type RM Length L Ch R = 1 ,47102.3 ,293.2,300,308.4
XS GIS Cut Line= 3
     1989325.858      322063.677     1989621.851       322536.53
     1989935.512      322980.887
#Sta/Elev= 30
       0 2718.07      10 2714.08    29.9 2705.39    99.6  2672.5   159.4  2645.2
   199.2 2626.44     249 2604.21   298.8 2582.69   328.7 2570.48   408.4 2539.73
   438.3 2528.94   458.2 2520.23   498.1  2501.1     518 2491.37   537.9 2480.78
   547.9 2478.02   550.4 2477.97   557.8 2477.81   565.4 2478.68   617.2 2486.03
   696.3 2496.17   706.2 2497.78     726 2502.61   864.4  2539.6   874.3 2542.61
     904 2552.85  1032.5 2598.47  1042.4 2602.31  1052.3  2606.6  1101.8 2629.11
#Mann= 3 , 0 , 0
       0      .1       0   550.4    .045       0   565.4      .1       0
Bank Sta=550.4,565.4
XS Rating Curve= 0 ,0
Exp/Cntr=0.3,0.1

Type RM Length L Ch R = 1 ,46802.3 ,603.6,599.7,594
XS GIS Cut Line= 3
     1989201.719      322111.244     1989342.732      322640.041
     1989475.186      323170.919
#Sta/Elev= 30
       0  2758.5    49.8 2736.11    89.6 2716.79   129.4 2693.85   169.2 2672.06
   189.1 2660.79   268.7 2614.02   328.4 2577.45   338.3 2570.76   358.2 2555.62
   368.2  2548.4   378.1 2542.77   417.9 2525.96   457.7  2507.4   497.5 2491.45
   507.5 2487.12   517.4 2481.99   527.4 2477.43   537.3 2475.24   539.8 2475.22
   547.3 2475.16   554.8  2475.8   656.7 2485.88   686.6 2489.31   805.9 2509.03
   835.8 2514.74   945.2 2537.74     995 2546.61  1054.6 2560.57  1094.4 2568.37
#Mann= 3 , 0 , 0
       0      .1       0   539.8    .045       0   554.8      .1       0
Bank Sta=539.8,554.8
XS Rating Curve= 0 ,0
Exp/Cntr=0.3,0.1

Type RM Length L Ch R = 1 ,46202.3 ,260.2,255.3,250.4
XS GIS Cut Line= 3
     1988560.094      322362.488     1988789.212      322856.055
      1989055.34      323344.577
#Sta/Elev= 30
       0 2744.74      89 2716.47   118.7 2703.56   158.3  2683.2   168.2 2675.25
     188 2656.71   197.9 2648.58   296.8 2578.07   306.7 2569.42   326.5 2548.35
   336.4 2538.94   346.3  2533.3   366.1 2528.35   395.8 2527.75   405.6 2526.59
   415.5 2523.71   474.9 2496.21   536.7 2474.16   544.2    2472   551.7 2471.45
   554.1 2471.28     564 2472.09   603.8 2478.69   623.6 2480.58   792.5  2484.9
     872 2495.57   911.7 2502.84  1001.1 2522.69    1021 2529.04  1100.5 2559.27
#Mann= 3 , 0 , 0
       0      .1       0   536.7    .045       0   551.7      .1       0
Bank Sta=536.7,551.7
XS Rating Curve= 0 ,0
Exp/Cntr=0.3,0.1

Type RM Length L Ch R = 1 ,45947   ,333.9,344.6,357.6
XS GIS Cut Line= 3
     1988256.639      322578.314     1988588.813      323012.183
     1988950.639      323424.893
#Sta/Elev= 30
       0 2756.89    29.8 2750.95   129.2 2715.89     159 2703.22   188.8 2686.41
   198.7 2678.92   218.6 2660.17   258.3 2616.72   268.2 2606.96   327.9 2559.04
   377.5  2516.1   387.5 2510.68   397.4 2508.32   427.2 2507.72   437.1 2505.89
   506.7 2480.53   526.6 2472.06   537.8 2469.22   546.4 2468.88   552.8 2470.12
   576.4 2477.22   586.3 2478.87   716.1 2487.75   795.9 2487.95   815.9 2489.68
   855.8 2498.81   935.6 2512.44   965.6 2519.02   995.5 2529.03  1095.3 2566.05
#Mann= 3 , 0 , 0
       0      .1       0   537.8    .045       0   552.8      .1       0
Bank Sta=537.8,552.8
XS Rating Curve= 0 ,0
Exp/Cntr=0.3,0.1

Type RM Length L Ch R = 1 ,45602.3 ,377.9,384.3,389.8
XS GIS Cut Line= 3
     1988242.546      322719.728     1988331.793      323198.926
     1988399.302       323678.98
#Sta/Elev= 30
       0 2716.71    19.9 2710.78    39.8 2703.66    49.7 2699.43    59.7 2694.52
    69.6 2688.28    79.6 2680.38   109.4 2654.34   149.2 2620.79   169.1 2604.77
   288.5 2516.32   298.4 2509.18   308.4 2503.38   318.3 2499.63   328.3 2497.21
   479.9 2464.08   487.4 2462.88   494.9 2462.64   497.3 2462.56   507.2 2463.27
   576.5 2472.42   596.3 2474.09     626 2476.03   645.7 2477.91   774.4 2493.89
   794.1 2496.59     804 2498.62   813.9  2501.6   853.5 2515.54   972.2 2558.78
#Mann= 3 , 0 , 0
       0      .1       0   479.9    .045       0   494.9      .1       0
Bank Sta=479.9,494.9
XS Rating Curve= 0 ,0
Exp/Cntr=0.3,0.1

Type RM Length L Ch R = 1 ,45218   ,221,221.1,222.5
XS GIS Cut Line= 2
     1988017.941      322661.237     1987910.317      323721.094
#Sta/Elev= 30
       0 2712.01    69.7 2679.59    99.6 2663.13   119.5 2649.55   159.3 2620.72
     219 2580.72   278.8  2542.4   298.7 2530.81   328.6 2517.94   388.3  2494.3
   487.8 2461.99   497.8 2459.59   507.8 2459.13   512.8 2459.34   627.2 2466.76
   647.2  2471.7     687 2486.02   696.9 2488.15   716.8 2489.71   746.7 2495.09
   766.6  2497.2   826.4 2500.22   836.3 2499.79   846.3 2497.33   866.2 2489.49
   876.1 2489.15     896 2494.35   935.9 2508.85   945.8 2511.56  1065.3  2526.2
#Mann= 3 , 0 , 0
       0      .1       0   497.8    .045       0   512.8      .1       0
Bank Sta=497.8,512.8
XS Rating Curve= 0 ,0
Exp/Cntr=0.3,0.1

Type RM Length L Ch R = 1 ,44996.8 ,298.8,294.4,287.4
XS GIS Cut Line= 3
     1987807.758      322614.868     1987748.882      323164.259
     1987658.953      323701.189
#Sta/Elev= 30
       0 2689.72    29.6 2669.53   108.5 2617.63   138.1 2599.16   167.7 2581.76
   197.3 2565.43     296 2519.41   335.5 2504.44   365.1  2496.3   434.1 2481.14
   544.3 2459.28   552.5 2458.59   559.3 2458.93   621.8 2467.83   681.2 2480.75
   720.8 2488.46   730.7 2489.42     800 2491.96   859.4 2495.84   889.1 2496.92
     899  2496.8   908.9 2495.53   948.5 2485.79   978.2 2479.77   988.1 2478.99
  1007.9 2482.26  1027.7 2482.04  1037.6 2483.77  1047.4 2488.15    1097 2515.77
#Mann= 3 , 0 , 0
       0      .1       0   544.3    .045       0   559.3      .1       0
Bank Sta=544.3,559.3
XS Rating Curve= 0 ,0
Exp/Cntr=0.3,0.1

Type RM Length L Ch R = 1 ,44702.3 ,239.8,237.1,236.9
XS GIS Cut Line= 4
     1987452.799      322626.098      1987437.71      322855.427
      1987461.59       323124.62     1987543.998      323688.801
#Sta/Elev= 30
       0 2605.99      60  2583.9    79.9 2574.67   129.9 2554.03   149.9 2543.55
   209.8  2509.5   219.8 2504.38   229.8 2500.69   239.8 2498.99   289.9 2495.78
   309.9 2493.12     470 2461.38   492.6 2458.33   500.1  2458.2   507.6  2458.4
   640.1  2463.2   660.1 2466.26   720.1 2479.72   750.2 2484.13   770.2 2485.57
   870.2 2485.96   920.2 2482.87   940.2 2479.11   950.2 2478.32   980.2 2483.95
  1000.2 2481.72  1010.2 2481.88  1020.2 2486.04  1050.2 2506.84  1070.2  2519.6
#Mann= 3 , 0 , 0
       0      .1       0   492.6    .045       0   507.6      .1       0
Bank Sta=492.6,507.6
XS Rating Curve= 0 ,0
Exp/Cntr=0.3,0.1

Type RM Length L Ch R = 1 ,44464.9 ,693.5,713.2,732.2
XS GIS Cut Line= 6
      1987187.75      322714.447     1987192.048      322890.521
     1987215.444      323065.994     1987264.576        323290.6
      1987309.03      323590.074     1987379.219      323987.813
#Sta/Elev= 30
       0 2591.45    19.6 2585.19    39.1  2577.2   117.4 2540.19     137 2528.92
   166.3 2508.09   176.1 2502.03     186 2498.36   195.8 2497.05   264.6 2494.17
   373.2 2465.34   433.1 2459.09   450.3  2458.2   453.1 2458.14   465.3 2458.24
   553.1 2461.34   563.1 2463.55   602.6 2478.32   612.4 2480.83   631.9 2483.18
   719.8 2484.84   827.2 2482.56   925.2 2484.24   935.1 2485.77   944.9 2490.14
   994.2 2520.17  1013.9 2530.33  1092.7 2562.28  1220.8 2619.86  1289.7 2647.06
#Mann= 3 , 0 , 0
       0      .1       0   450.3    .045       0   465.3      .1       0
Bank Sta=450.3,465.3
XS Rating Curve= 0 ,0
Exp/Cntr=0.3,0.1

Type RM Length L Ch R = 1 ,43751.2 ,529.9,548,566.9
XS GIS Cut Line= 5
     1987121.488      322696.041     1987042.311      322853.087
     1986887.894      323063.655     1986483.037      323573.138
     1986384.871      323693.018
#Sta/Elev= 30
       0 2593.05    39.1 2582.03    68.4 2571.09    87.9 2562.37   146.6 2533.72
   195.2 2502.36   204.9 2497.21   214.6 2495.31   282.3 2492.65   301.6 2488.07
   388.6 2462.78   415.8 2458.02   430.8 2457.95     467 2457.82   587.2 2458.36
   687.3 2460.56   697.3  2462.1   757.4 2482.26   777.4 2485.19   857.5 2483.32
   897.5 2484.72   967.6 2477.59   987.6 2478.28  1007.7 2480.66  1027.7  2486.6
  1057.7 2502.37  1107.1 2525.93  1136.2 2543.59  1165.2 2559.28  1242.7 2595.07
#Mann= 3 , 0 , 0
       0      .1       0   415.8    .045       0   430.8      .1       0
Bank Sta=415.8,430.8
XS Rating Curve= 0 ,0
Exp/Cntr=0.3,0.1

Type RM Length L Ch R = 1 ,43202.3 ,295.1,300.1,303.7
XS GIS Cut Line= 4
     1987063.367      322710.369     1986808.346      322846.068
     1986589.408      322877.502     1986098.039      322919.954
#Sta/Elev= 30
       0 2579.59      10 2575.91    29.9 2567.01    79.7 2541.59    99.6 2530.69
   139.5 2504.89   149.4 2499.08   159.4 2495.81   209.2  2496.7   219.2 2496.52
   229.1 2495.35   288.9 2480.35   365.8 2462.44     385  2461.1   500.4 2457.94
   502.6 2457.94   517.6 2458.34     589 2465.45   598.8 2467.93   608.7    2472
   638.3 2486.52   648.2  2490.1     658 2491.42   796.1 2488.25     806 2488.24
   815.8 2489.59   825.7 2492.94   944.1 2544.55   963.8 2551.99  1003.3    2565
#Mann= 3 , 0 , 0
       0      .1       0   502.6    .045       0   517.6      .1       0
Bank Sta=502.6,517.6
XS Rating Curve= 0 ,0
Exp/Cntr=0.3,0.1

Type RM Length L Ch R = 1 ,42902.3 ,325.7,327.9,330.2
XS GIS Cut Line= 4
     1987084.424       322572.33     1986930.008      322593.387
     1986626.108      322587.578     1986103.108      322579.587
#Sta/Elev= 30
       0 2594.78     9.7 2588.88    29.2 2578.63   116.9 2538.54   126.6    2532
   136.4 2523.28   155.8 2503.22   165.6 2495.56   175.5 2492.53   253.9 2490.67
   273.5 2489.51   283.3 2487.71   391.2 2461.55     401 2460.38   452.3 2458.01
   459.8 2457.96   467.3 2458.93   469.7 2459.24   499.3 2468.35   528.9 2475.52
   627.6 2496.46   657.2 2500.62   676.9 2501.98   706.5 2499.51   716.4 2500.22
   726.3 2503.86   834.8 2568.67     894 2603.33   963.1  2642.7   982.9 2652.99
#Mann= 3 , 0 , 0
       0      .1       0   452.3    .045       0   467.3      .1       0
Bank Sta=452.3,467.3
XS Rating Curve= 0 ,0
Exp/Cntr=0.3,0.1

Type RM Length L Ch R = 1 ,42574.1 ,257.6,256,254.5
XS GIS Cut Line= 2
     1987332.978      322406.999     1986204.719      322235.422
#Sta/Elev= 30
       0 2661.64      20  2658.6      40 2652.62    70.1 2641.12   110.1 2623.56
   180.2 2590.56   250.3 2558.64   260.3 2553.14   330.4 2509.97   340.4 2504.44
   350.4 2500.79   360.4 2499.28   430.5 2495.79   450.5 2492.86   560.2 2457.98
   575.2 2456.85   580.6 2456.84   650.7 2457.42   670.7 2458.63   690.8  2464.4
   780.8 2497.19   800.9 2503.17   810.9 2504.22     901 2506.48     921 2505.83
   981.1 2501.54   991.1 2503.21  1011.1  2511.1  1091.2 2546.13  1141.2 2565.27
#Mann= 3 , 0 , 0
       0      .1       0   560.2    .045       0   575.2      .1       0
Bank Sta=560.2,575.2
XS Rating Curve= 0 ,0
Exp/Cntr=0.3,0.1

Type RM Length L Ch R = 1 ,42318   ,624.3,614.8,601.2
XS GIS Cut Line= 4
     1987482.163      322132.478     1986890.234      322083.345
     1986665.641      322064.182     1986234.859      322062.227
#Sta/Elev= 30
       0 2637.19      99 2614.73   237.6 2569.28   257.4 2560.64   267.3 2555.11
   336.6 2509.57   346.5  2504.7   356.4 2501.71   366.3 2500.48   386.1 2500.44
   475.2 2503.74     495 2503.15   514.8 2498.35   544.5 2488.52     627 2458.01
   633.2  2456.8     642 2456.81   721.4 2458.07     790 2462.52   887.9 2473.77
   936.9 2480.95   985.8 2485.61  1044.6 2495.99  1093.5  2509.6  1103.3  2510.6
  1142.5 2510.67    1211 2508.28  1220.8  2509.3  1230.6    2512  1250.2 2520.65
#Mann= 3 , 0 , 0
       0      .1       0     627    .045       0     642      .1       0
Bank Sta=627,642
XS Rating Curve= 0 ,0
Exp/Cntr=0.3,0.1

Type RM Length L Ch R = 1 ,41702.3 ,313.4,299.6,266.8
XS GIS Cut Line= 4
     1987185.056      321262.894     1986939.366      321545.228
      1986802.78      321620.935     1986181.323      322013.156
#Sta/Elev= 30
       0 2583.94    49.2 2542.24    78.8  2518.6    88.6  2512.8    98.5 2509.36
   108.3 2508.15   137.9 2507.64   246.2 2509.18   265.9  2508.3   295.5 2500.66
   374.3 2476.13   403.6 2468.87   462.1 2457.77   522.9 2455.65   530.4  2455.5
   537.9 2455.68   768.8 2462.19   828.4 2465.43   868.1  2469.2   907.8 2474.44
   997.2 2489.93    1017 2496.56  1046.8 2508.89  1066.7 2514.18  1116.4 2515.13
  1175.9 2509.87  1205.7 2509.05  1215.7 2511.67  1225.6  2516.9  1265.3 2544.12
#Mann= 3 , 0 , 0
       0      .1       0   522.9    .045       0   537.9      .1       0
Bank Sta=522.9,537.9
XS Rating Curve= 0 ,0
Exp/Cntr=0.3,0.1

Type RM Length L Ch R = 1 ,41402.3 ,304.3,300,321.7
XS GIS Cut Line= 3
     1987060.854      321135.254     1986607.889      321473.164
     1986168.537       321888.81
#Sta/Elev= 30
       0 2609.02    39.7 2589.71    59.5 2577.11    89.2 2556.36    99.1 2550.31
   109.1 2545.47     119 2543.02   148.7 2541.99     238 2527.23   267.7 2518.67
   297.4 2508.29   337.1 2497.72   436.2 2463.24   456.1 2457.86   505.6 2454.58
   557.6 2453.01   565.1 2452.92   572.6 2452.95   654.4 2457.36   773.3  2460.1
   872.5 2463.99   892.3 2467.47   991.5    2506  1001.4 2509.42  1021.2 2514.22
    1041 2516.28  1070.8 2516.59  1150.1 2512.86    1160 2513.57  1169.9 2516.35
#Mann= 3 , 0 , 0
       0      .1       0   557.6    .045       0   572.6      .1       0
Bank Sta=557.6,572.6
XS Rating Curve= 0 ,0
Exp/Cntr=0.3,0.1

Type RM Length L Ch R = 1 ,41102.3 ,293.6,299.9,300.7
XS GIS Cut Line= 3
      1986531.29      320809.156     1986393.513       321328.47
     1986104.314      321848.934
#Sta/Elev= 30
       0 2597.81    69.6  2551.9    89.6 2541.18   139.3  2517.7   149.2 2515.72
   159.2 2515.62   268.6 2519.61   278.6 2519.81   288.5 2519.23   298.5 2517.29
   308.4  2514.2   457.7 2462.24   467.6 2459.75   477.6 2458.38   507.4 2456.05
   529.8 2452.92   537.3 2452.42   544.8 2452.48   785.4 2461.96   795.3 2463.59
   805.2 2466.24   894.5 2498.05   924.3 2507.75   944.2 2513.44   954.1 2515.07
     964 2515.28  1102.9 2513.06  1112.8  2513.9  1122.8 2517.48  1132.7 2523.77
#Mann= 3 , 0 , 0
       0      .1       0   529.8    .045       0   544.8      .1       0
Bank Sta=529.8,544.8
XS Rating Curve= 0 ,0
Exp/Cntr=0.3,0.1

Type RM Length L Ch R = 1 ,40802.1 ,300.7,299.7,299.3
XS GIS Cut Line= 3
     1986411.333      320765.272     1986039.794      321377.548
     1985764.482      321661.038
#Sta/Elev= 30
       0 2605.76    49.7 2571.99    89.5 2547.67   109.4 2538.55   169.1 2518.48
     179 2515.94     189 2514.58   298.4 2517.03   318.3 2515.56     368 2501.15
   387.9 2493.97   447.6 2470.13   477.5 2460.98   497.4 2456.81   517.2 2454.27
   572.4  2451.9   586.9  2451.5   587.4 2451.51   606.8 2452.69   795.2 2482.75
     815 2488.55   854.5 2506.19   864.4 2509.08   953.3 2518.47  1002.7 2516.03
  1012.6 2515.92  1022.4 2517.29  1032.3 2521.08    1062 2535.99  1111.4 2567.13
#Mann= 3 , 0 , 0
       0      .1       0   572.4    .045       0   587.4      .1       0
Bank Sta=572.4,587.4
XS Rating Curve= 0 ,0
Exp/Cntr=0.3,0.1

Type RM Length L Ch R = 1 ,40502.3 ,295.3,300,303.7
XS GIS Cut Line= 3
     1986142.154       320604.82     1985881.773      321084.431
      1985609.51      321558.574
#Sta/Elev= 30
       0  2643.1    29.8 2622.95    69.5  2594.5    89.3 2581.76   119.1 2565.54
   158.8 2548.16     258 2512.42   267.9 2510.42   277.8  2510.4   337.4 2516.64
   347.3 2516.64   357.2 2514.91   466.4 2473.59     516  2452.7   525.9 2451.28
   538.2 2451.86   553.2 2453.47     675  2466.1   744.6 2475.99   754.5 2477.96
   764.4 2481.18   814.1 2502.67     834 2508.97     844  2510.8   903.6  2513.7
   943.4 2518.96    1013 2523.17  1022.9 2525.62  1032.8 2530.16  1092.5 2565.07
#Mann= 3 , 0 , 0
       0      .1       0   538.2    .045       0   553.2      .1       0
Bank Sta=538.2,553.2
XS Rating Curve= 0 ,0
Exp/Cntr=0.3,0.1

Type RM Length L Ch R = 1 ,40202.3 ,309.9,300,293.6
XS GIS Cut Line= 3
     1985980.369      320517.091       1985622.1      320937.428
     1985277.057      321359.148
#Sta/Elev= 30
       0 2637.34    88.8 2572.17    98.6  2565.7   118.4 2556.73   246.6 2507.05
   256.4 2505.38   266.3 2505.13   345.2 2505.66   374.8 2505.05   384.6 2503.77
     503 2465.16   532.6 2454.35   544.8 2451.32   552.3 2450.57   559.8 2450.91
   710.8 2465.01   720.7 2466.58   730.6 2469.13   809.9 2495.03   839.6 2503.24
   859.4 2507.71   918.9 2516.05   928.8 2516.76   968.4 2515.63  1017.9 2522.11
  1027.8 2522.88  1047.7 2522.84  1057.6 2524.37  1067.5 2528.07  1097.2 2542.68
#Mann= 3 , 0 , 0
       0      .1       0   544.8    .045       0   559.8      .1       0
Bank Sta=544.8,559.8
XS Rating Curve= 0 ,0
Exp/Cntr=0.3,0.1
